--- J100-00-00.prj (project) ---

Proj Title=J100-00-00
Current Plan=p01
Default Exp/Contr=.3,.1
English Units
Geom File=g01
Flow File=f02
Flow File=f01
Plan File=p02
Plan File=p01
Y Axis Title=Elevation
X Axis Title(PF)=Main Channel Distance
X Axis Title(XS)=Station
BEGIN DESCRIPTION:
HCFCD Watershed Unit ID: J
M3 Study Identifier: 2007_Effective_J
Engineer: HCFCD
Project Name: Effective FEMA Study for watershed Spring Creek (J)
Study Completion Date: 6/18/2007
FEMA Case Number: [No Data]
FEMA Approval Date: [No Date in Database]
Vertical Datum: NAVD 1988
Datum Note: 2001 ADJ
HYDRAULICS
HCFCD Unit No.:  J100-00-00
Hydraulic Program Name: HEC-RAS
Hydraulic Program Version: 3.0.1
Steady Hydraulic Model: Yes
Unsteady Hydraulic Model: No
Update 1:
The effective FEMA hydraulic model for unit number J100-00-00 has been updated by FEMA LOMR 09-06-1932P with an effective date of 6/26/2009.
Update 2:
The effective FEMA hydraulic model for unit number J100-00-00 has been updated by FEMA LOMR 14-06-1656P with an effective date of 10/03/2014.
END DESCRIPTION:
DSS Export Rating Curves= 0
DSS Export Rating Curve Sorted= 0
DSS Export Volume Flow Curves= 0
DXF OffsetX= 0
DXF OffsetY= 0
DXF ScaleX= 1
DXF ScaleY= 10

--- J100-00-00.p01 (plan) ---

Plan Title=FEMA Effective Multi-Profile 2014
Version=Version 3.0.1  May 2012
Short Identifier=Eff+LOMR MP
Geom File=g01
Flow File=f01
Subcritical Flow
K Sum by GR= 0
Std Step Tol= 0.01
Critical Tol= 0.01
Num of Std Step Trials= 20
Max Error Tol= 0.3
Flow Tol Ratio= 0.001
Split Flow NTrial= 30
Split Flow Tol= 0.02
Split Flow Ratio= 0.02
Log Output Level= 0
Friction Slope Method= 1
Unsteady Friction Slope Method= 2
Parabolic Critical Depth
Global Vel Dist= 0 , 0 , 0
Global Log Level= 0
CheckData=True
Encroach Param=-1 ,0,0, 0
BEGIN DESCRIPTION:
FEMA Effective June 2007 +...+ LOMR 14-06-1656P
END DESCRIPTION:
Computation Interval=1HOUR
Output Interval=1HOUR
Run HTab= 0
Run UNet= 0
Run PostProcess= 0
UNET Theta= 1
UNET ZTol= 0.02
UNET ZSATol= 0.1
UNET MxIter= 20
UNET MaxInSteps= 20
UNET DtIC= 0
UNET DtMin= 0
UNET MaxCRTS= 20
UNET WFStab= 2
UNET SFStab= 1
UNET WFX= 1
UNET SFX= 1
UNET Convert EG Bridges=-1
UNET Use Existing IB Tables=-1
Instantaneous Interval=1HOUR
Write IC File= 0
Write Velocity= 0
Write Detailed= 0

--- J100-00-00.p02 (plan) ---

Plan Title=FEMA Effective Floodway 2014
Version=Version 3.0.1  May 2012
Short Identifier=Eff+LOMR FW
Geom File=g01
Flow File=f02
Subcritical Flow
K Sum by GR= 0
Std Step Tol= 0.01
Critical Tol= 0.01
Num of Std Step Trials= 20
Max Error Tol= 0.3
Flow Tol Ratio= 0.001
Split Flow NTrial= 30
Split Flow Tol= 0.02
Split Flow Ratio= 0.02
Log Output Level= 0
Friction Slope Method= 1
Unsteady Friction Slope Method= 2
Parabolic Critical Depth
Global Vel Dist= 0 , 0 , 0
Global Log Level= 0
CheckData=True
Encroach Param=-1 ,0,0, 2
Encroach River=J100-00-00
Encroach Reach=Reach - 1
Encroach Node=367736.2
       1    4895    5050
Encroach Node=367286.5
       1    4985    5325
Encroach Node=366730.7
       1    4985    5165
Encroach Node=366583.5
       1    4950    5160
Encroach Node=366558.0
       1    4950    5160
Encroach Node=366532.5
       1    4950    5160
Encroach Node=366281.2
       1    4945    5202
Encroach Node=365737.8
       1    4935    5084
Encroach Node=365177.7
       1    4955    5085
Encroach Node=364609.2
       1    4975    5020
Encroach Node=363767.8
       1    4965    5035
Encroach Node=362623.4
       1    4970    5350
Encroach Node=361421.5
       1    4985    5285
Encroach Node=360650.7
       1    4700    5217
Encroach Node=359656.4
       1    4895    5260
Encroach Node=358871.8
       1    4915    5025
Encroach Node=358760
       1  4959.6  5049.5
Encroach Node=358711.9
       1  4959.6  5049.5
Encroach Node=358670
       1  4959.6  5049.5
Encroach Node=358431.6
       1    4955    5220
Encroach Node=357927.6
       1    4985    5280
Encroach Node=356334.4
       1    4530    5060
Encroach Node=355818.6
       1    4560    5015
Encroach Node=355803.6
       1    4560    5015
Encroach Node=355788.6
       1    4560    5015
Encroach Node=355220.5
       1    4850    5305
Encroach Node=354502.3
       1    4610    5020
Encroach Node=353146.4
       1    4380    5020
Encroach Node=352519.9
       1    4865    5485
Encroach Node=352448.5
       1    4895    5520
Encroach Node=352431.5
       1    4895    5520
Encroach Node=352414.5
       1    4895    5520
Encroach Node=352094.8
       1    4730    5480
Encroach Node=351184.1
       1    4700    5195
Encroach Node=349666.6
       1    4980    5715
Encroach Node=348410.9
       1    4525    5020
Encroach Node=347486.7
       1    4964    5614
Encroach Node=346570.3
       1    4650    5020
Encroach Node=344901.6
       1    4368    5073
Encroach Node=343432.7
       1    4520    5016
Encroach Node=342134.8
       1    4779    5340
Encroach Node=341654.0
       1    4875    5345
Encroach Node=340883.3
       1    4455    5045
Encroach Node=340800.4
       1    4455    5300
Encroach Node=340768.9
       1    4455    5300
Encroach Node=340737.4
       1    4455    5300
Encroach Node=340480.0
       1    4590    5365
Encroach Node=339806.4
       1    4510    5395
Encroach Node=338783.3
       1    4810    5490
Encroach Node=337922.3
       1    4067    5021
Encroach Node=337168.3
       1    3813    5058
Encroach Node=335710.7
       1    4000    5240
Encroach Node=333741.8
       1    4400    5020
Encroach Node=333114.7
       1    4255    5025
Encroach Node=332505.1
       1    3865    5015
Encroach Node=332186.3
       1    3945    5050
Encroach Node=331980.1
       1    3950    5050
Encroach Node=331810
       1    3920    5030
Encroach Node=331768
       1    3920    5030
Encroach Node=331726
       1    3920    5030
Encroach Node=331580.1
       1    3875    5040
Encroach Node=331161.5
       1    3850    5170
Encroach Node=329870.1
       1    4645    5700
Encroach Node=329103.9
       1    4622    5593
Encroach Node=327680.9
       1    3920    5075
Encroach Node=326067.5
       1    4980    5870
Encroach Node=324978.2
       1    4735    5510
Encroach Node=324699.3
       1    4640    5395
Encroach Node=324675.3
       1    4640    5395
Encroach Node=324651.3
       1    4640    5395
Encroach Node=324448.5
       1    4665    5430
Encroach Node=324126.4
       1    4710    5450
Encroach Node=322581.7
       1    4930    6005
Encroach Node=322049.6
       1    4980    5510
Encroach Node=320841.0
       1    4678    5163
Encroach Node=319539.7
       1    4980    5305
Encroach Node=318256.3
       1    4699    5249
Encroach Node=317377.2
       1    4980    5435
Encroach Node=316442.7
       1    4680    5790
Encroach Node=314695.6
       1    4555    5035
Encroach Node=314083.9
       1    4530    5075
Encroach Node=313747.7
       1    4630    5080
Encroach Node=313556.0
       1    4530    5060
Encroach Node=313528.0
       1    4530    5060
Encroach Node=313500.0
       1    4530    5060
Encroach Node=313379.2
       1    4485    5030
Encroach Node=312917.5
       1    4560    5040
Encroach Node=312109.2
       1    4450    5170
Encroach Node=310620.7
       1    4740    5080
Encroach Node=309811.2
       1    4628    5032
Encroach Node=308858.1
       1    4975    5335
Encroach Node=308143.7
       1    4159    5066
Encroach Node=307032.4
       1    4885    5430
Encroach Node=306637.5
       1    4935    5240
Encroach Node=305929.2
       1    4855    5240
Encroach Node=305093.2
       1    4925    5280
Encroach Node=304581.5
       1    4840    5200
Encroach Node=303924.9
       1    4843    5145
Encroach Node=303573.5
       1    4880    5200
Encroach Node=303021.8
       1    4674    5116
Encroach Node=301168.9
       1    4700    5110
Encroach Node=300789.3
       1    4650    5430
Encroach Node=300588.4
       1    4290    5080
Encroach Node=300563.4
       1    4290    5080
Encroach Node=300538.4
       1    4290    5080
Encroach Node=300417.1
       1    4600    5450
Encroach Node=300206.7
       1    4600    5450
Encroach Node=299727.1
       1    4495    5425
Encroach Node=298613.9
       1    4235    5020
Encroach Node=296972.1
       1    4930    5370
Encroach Node=295216.8
       1  3673.5    5095
Encroach Node=293785.3
       1    4265    5040
Encroach Node=292719.4
       1    4500    5240
Encroach Node=291773.9
       1    4800    5365
Encroach Node=290617.0
       1    4370    5010
Encroach Node=289038.3
       1    4977    5630
Encroach Node=288387.2
       1    4910    5535
Encroach Node=288254.7
       1    4880    5595
Encroach Node=288228.7
       1    4880    5595
Encroach Node=288202.7
       1    4880    5595
Encroach Node=288101.9
       1    4820    5500
Encroach Node=287629.8
       1    4808    5451
Encroach Node=286810.8
       1    4340    5025
Encroach Node=286019.2
       1    4780    5390
Encroach Node=285474.5
       1    4820    5505
Encroach Node=284884.7
       1    4840    5425
Encroach Node=284224.5
       1    4779    5414
Encroach Node=283056.7
       1    4560    5135
Encroach Node=281683.2
       1    4250    5150
Encroach Node=281325.9
       1    4000    5350
Encroach Node=281309.9
       1    4000    5350
Encroach Node=281293.9
       1    4000    5350
Encroach Node=281230.1
       1    4000    5400
Encroach Node=280415.4
       1    4300    5240
Encroach Node=279957.0
       1    4685    5420
Encroach Node=278974.0
       1    4205    5500
Encroach Node=276574.0
       1    4570    6110
Encroach Node=275250.8
       1    4410    5460
Encroach Node=274419.1
       1    4725    5555
Encroach Node=273050.2
       1    4619    5165
Encroach Node=271847.4
       1    4401    5024
Encroach Node=270264.8
       1    4550    5566
Encroach Node=268978.8
       1    4113    5057
Encroach Node=268443.6
       1    4259    5069
Encroach Node=267069.3
       1    4922    5663
Encroach Node=266006.8
       1    4578    5564
Encroach Node=265776.4
       1    4555    5485
Encroach Node=265745.1
       1    4555    5485
Encroach Node=265713.9
       1    4555    5485
Encroach Node=265483.0
       1    4301    5381
Encroach Node=265026.2
       1    4002    5048
Encroach Node=264692.5
       1    3930    5078
Encroach Node=263211.6
       1    4511    5441
Encroach Node=262727.2
       1    4703    5487
Encroach Node=261953.2
       1    4380    5158
Encroach Node=260953.0
       1    4885    5411
Encroach Node=260773.2
       1    4930    5439
Encroach Node=260537.4
       1    4935    5441
Encroach Node=260505.9
       1    4935    5441
Encroach Node=260474.4
       1    4935    5441
Encroach Node=260390.6
       1    4850    5392
Encroach Node=260014.0
       1    4683    5178
Encroach Node=259563.8
       1    4582    5040
Encroach Node=258009.9
       1    4403    5554
Encroach Node=257100.6
       1    4170    5163
Encroach Node=255371.0
       1    4707    5568
Encroach Node=254627.6
       1    4925    5615
Encroach Node=253915.9
       1    4400    5376
Encroach Node=253565.0
       1    4095    5200
Encroach Node=253257.0
       1    3850    5065
Encroach Node=253220.0
       1    3850    5065
Encroach Node=253183.0
       1    3850    5065
Encroach Node=253055.3
       1    3593    5065
Encroach Node=252295.8
       1    3640    5175
Encroach Node=250563.3
       1    3945    5450
Encroach Node=249516.8
       1    4125    5565
Encroach Node=247895.6
       1    4704    6150
Encroach Node=246746.6
       1    4580    5835
Encroach Node=244790.2
       1    4350    5600
Encroach Node=243422.6
       1    3846    5136
Encroach Node=242215.8
       1    4830    6150
Encroach Node=241149.2
       1    4870    6150
Encroach Node=239561.0
       1  4272.2    5290
Encroach Node=239260.1
       1    4080    5160
Encroach Node=239229.6
       1    4080    5160
Encroach Node=239199.1
       1    4080    5160
Encroach Node=238748.0
       1    3918    5069
Encroach Node=237861.9
       1    4000    5200
Encroach Node=236547.8
       1    4056    5305
Encroach Node=235332.5
       1    3390    5080
Encroach Node=234734.7
       1    3370  5041.8
Encroach Node=233292.2
       1    3270    5680
Encroach Node=230694.7
       1    3803    6925
Encroach Node=229710.8
       1    4065    6745
Encroach Node=228588.3
       1    3640    6025
Encroach Node=227253.1
       1    2250    5297
Encroach Node=225153.4
       1    1305    5040
Encroach Node=223808.7
       1    1390    5155
Encroach Node=221840.8
       1    2832    6385
Encroach Node=221103.6
       1    3400    6230
Encroach Node=219902.0
       1    3450    5515
Encroach Node=217354.5
       1  4309.8  6359.3
Encroach Node=213918.9
       1    2740    5200
Encroach Node=211631.6
       1    3300    5250
Encroach Node=210431.1
       1    3850    5600
Encroach Node=209190.3
       1    4260    5905
Encroach Node=208249.9
       1    4510    6005
Encroach Node=207799.6
       1  4212.5    6065
Encroach Node=207518.1
       1    3650    5900
Encroach Node=207453.1
       1    3650    5900
Encroach Node=207388.1
       1    3650    5900
Encroach Node=207139.4
       1    3621    5800
Encroach Node=206325.6
       1    2745    5415
Encroach Node=205172.3
       1    2980    5140
Encroach Node=203889.5
       1    3515    5380
Encroach Node=202317.6
       1    3770    6170
Encroach Node=201301.7
       1    2835    5625
Encroach Node=199974.4
       1    2795    5040
Encroach Node=198833.4
       1    3575    5320
Encroach Node=198488.0
       1    3850    5300
Encroach Node=198318.6
       1    3850  5165.9
Encroach Node=198300.6
       1    3850  5165.9
Encroach Node=198282.6
       1    3850  5165.9
Encroach Node=198097.0
       1    3860    5450
Encroach Node=196302.3
       1    2625    5060
Encroach Node=193888.1
       1    3770    5550
Encroach Node=192987.0
       1    4300    6125
Encroach Node=192144.6
       1    4515    6480
Encroach Node=191675.8
       1    4664    6373
Encroach Node=190756.0
       1    4150  5325.7
Encroach Node=190739.5
       1    4150  5325.7
Encroach Node=190723.0
       1    4150  5325.7
Encroach Node=189712.6
       1    3950    5035
Encroach Node=188775.6
       1    3650    5090
Encroach Node=187576.7
       1    3250    5255
Encroach Node=186599.3
       1    4065    5600
Encroach Node=184626.4
       1    3085    5600
Encroach Node=182543.1
       1    3062    5030
Encroach Node=181868.6
       1    3700    5300
Encroach Node=181706.6
       1    3733    5385
Encroach Node=181671.6
       1    3733    5385
Encroach Node=181636.6
       1    3733    5385
Encroach Node=181281.7
       1    3500    5100
Encroach Node=180714.4
       1    3565    5280
Encroach Node=179254.7
       1    3330    5225
Encroach Node=177593.4
       1    3135    5085
Encroach Node=176206.0
       1    3257    5035
Encroach Node=174131.0
       1    3400    5495
Encroach Node=172966.9
       1    4280    6525
Encroach Node=171768.5
       1    4390    6731
Encroach Node=170367.7
       1    4460    7238
Encroach Node=168865.4
       1    4785    7475
Encroach Node=165536.3
       1    4743    7645
Encroach Node=163482.3
       1    4750    8040
Encroach Node=162164.1
       1    3850    7390
Encroach Node=159174.0
       1    2000    5617
Encroach Node=157651.2
       1    1975    5105
Encroach Node=156001.8
       1    3303    5340
Encroach Node=155042.3
       1    3070    5710
Encroach Node=153682.2
       1    4285    6670
Encroach Node=153142.6
       1    4175    6765
Encroach Node=151553.1
       1    3660    6400
Encroach Node=150642.0
       1    3335    5815
Encroach Node=149311.7
       1    4450    6470
Encroach Node=148935.1
       1    4629    6600
Encroach Node=148908.1
       1    4629    6600
Encroach Node=148881.1
       1    4629    6600
Encroach Node=148606.0
       1    4450    6210
Encroach Node=147849.6
       1    3700    5640
Encroach Node=146208.1
       1    3766    5560
Encroach Node=144510.7
       1    3335    5435
Encroach Node=141923.5
       1    4030    6036
Encroach Node=140963.4
       1    4080    6050
Encroach Node=139160.1
       1    3190    5320
Encroach Node=137656.0
       1    2675    5670
Encroach Node=136198.2
       1    3985    6045
Encroach Node=135401.0
       1    3850    5504
Encroach Node=134528.2
       1    4470    6125
Encroach Node=133785.6
       1    4215    5905
Encroach Node=131665.9
       1    4800    6125
Encroach Node=130131.1
       1    4315    6270
Encroach Node=129178.8
       1    4175    5765
Encroach Node=128719.4
       1 3983.69    5775
Encroach Node=128687.4
       1 3983.69    5775
Encroach Node=128636.7
       1 3983.69    5775
Encroach Node=128210.0
       1    4105    5675
Encroach Node=127566.0
       1    4190    6710
Encroach Node=126725.2
       1    3725    6475
Encroach Node=125593.6
       1    3675    6135
Encroach Node=124486.4
       1    3500  6432.1
Encroach Node=122390.6
       1    4160    6960
Encroach Node=121286.5
       1    4834    6950
Encroach Node=120290.5
       1    4345    6440
Encroach Node=117085.2
       1    3565    5616
Encroach Node=115715.2
       1    3400    6520
Encroach Node=114331.8
       1    4055    6590
Encroach Node=112909.9
       1    4350    6426
Encroach Node=110554.7
       1    3790    5850
Encroach Node=109165.1
       1    3530    5590
Encroach Node=107034.5
       1    3900    5875
Encroach Node=106148.0
       1    4300    6250
Encroach Node=104333.5
       1    3580    5880
Encroach Node=102794.9
       1    3770    5565
Encroach Node=100852.5
       1    3230    5120
Encroach Node=100361.0
       1    3092    5070
Encroach Node=99039.0
       1    3695    5649
Encroach Node=97170.6
       1    3720    6490
Encroach Node=95303.6
       1    3270    5940
Encroach Node=94465.9
       1  2717.4    5175
Encroach Node=93038.3
       1    3620    5310
Encroach Node=91780.8
       1    4275    5996
Encroach Node=90249.3
       1    4030    5750
Encroach Node=88797.0
       1    3575    5805
Encroach Node=88153.2
       1    3855    5790
Encroach Node=87559.3
       1    4055    5870
Encroach Node=87195.6
       1    3290    4835
Encroach Node=86927.5
       1    3290    4835
Encroach Node=86681.8
       1    3290    4835
Encroach Node=85856.6
       1    3745    5660
Encroach Node=84744.7
       1    3420    5890
Encroach Node=83099.6
       1    4160    6775
Encroach Node=82761.5
       1    4470    6975
Encroach Node=82743.3
       1    4470    6975
Encroach Node=82725.2
       1    4470    6975
Encroach Node=82073.8
       1    4765    7076
Encroach Node=80878.1
       1    4635    6495
Encroach Node=79447.2
       1    4225    6280
Encroach Node=78116.0
       1    3600    6705
Encroach Node=76553.3
       1    3170    5070
Encroach Node=76082.3
       1    3327    5070
Encroach Node=75018.5
       1    3780    5650
Encroach Node=73296.0
       1    4132    7019
Encroach Node=72547.7
       1    4786    6625
Encroach Node=71829.0
       1    4207    5813
Encroach Node=71348.7
       1    4150    5575
Encroach Node=70767.1
       1    4490    6035
Encroach Node=69737.8
       1    3580    5510
Encroach Node=69232.2
       1    3960    5760
Encroach Node=68984.0
       1    4110    5259
Encroach Node=68728.6
       1    3574    5362
Encroach Node=68706.1
       1    3574    5362
Encroach Node=68683.6
       1    3574    5362
Encroach Node=68507.9
       1    3640    5385
Encroach Node=68065.2
       1    3630    5750
Encroach Node=67818.7
       1    3660    5940
Encroach Node=67196.3
       1    3350    6200
Encroach Node=65844.4
       1    3110    6080
Encroach Node=64135.5
       1    2850    5505
Encroach Node=62959.6
       1    2618    5766
Encroach Node=61564.3
       1    2788    5810
Encroach Node=60210.3
       1    3540    5455
Encroach Node=58691.8
       1    4770    6500
Encroach Node=57733.4
       1    4625    6320
Encroach Node=56314.1
       1    4350    6545
Encroach Node=53962.3
       1    4680    6345
Encroach Node=52217.8
       1    4025    6625
Encroach Node=49773.6
       1    4153    5867
Encroach Node=48076.0
       1    4654    7162
Encroach Node=46243.5
       1    4430    6680
Encroach Node=45403.9
       1    4229    6445
Encroach Node=43924.4
       1    4625    6393
Encroach Node=42546.8
       1    3570    6190
Encroach Node=41576.1
       1    4300    6755
Encroach Node=40938.2
       1    4410    6900
Encroach Node=39313.9
       1    3340    6125
Encroach Node=36356.7
       1    2271    5100
Encroach Node=35047.8
       1    3450    5731
Encroach Node=34111.6
       1    3490    6110
Encroach Node=32535.7
       1    3000    5741
Encroach Node=31192.2
       1    2730    5440
Encroach Node=29692.8
       1    2500    5260
Encroach Node=29028.0
       1    2785    5070
Encroach Node=27592.1
       1    4500    5702
Encroach Node=26862.3
       1    4100    5585
Encroach Node=25883.5
       1    3100    5400
Encroach Node=24783.7
       1    2550    5315
Encroach Node=23405.3
       1    3045    5720
Encroach Node=22403.9
       1    4100    6030
Encroach Node=21505.6
       1    3750    5810
Encroach Node=20617.2
       1    3520    5865
Encroach Node=19133.4
       1    2917    6412
Encroach Node=17516.9
       1    3000    5520
Encroach Node=16413.7
       1    2390    5700
Encroach Node=15655.4
       1    2030    5254
Encroach Node=14080.8
       1    3320    6235
Encroach Node=13076.9
       1    3595    6120
Encroach Node=12248.6
       1    3635    6250
Encroach Node=10706.6
       1    4860    6550
Encroach Node=9272.5
       1  4365.5  5920.5
Encroach Node=8103.2
       1    4824    5692
Encroach Node=6876.4
       1    4684    5549
Encroach Node=5239.9
       1    3693    5372
Encroach Node=3019.7
       1    3557    6085
Encroach Reach=J100-00-00_0030
Encroach Node=367736.2
       1    4895    5050
Encroach Node=367286.5
       1    4985    5325
Encroach Node=366730.7
       1    4985    5165
Encroach Node=366583.5
       1    4950    5160
Encroach Node=366558.0
       1    4950    5160
Encroach Node=366532.5
       1    4950    5160
Encroach Node=366281.2
       1    4945    5202
Encroach Node=365737.8
       1    4935    5084
Encroach Node=365177.7
       1    4955    5085
Encroach Node=364609.2
       1    4975    5020
Encroach Node=363767.8
       1    4965    5035
Encroach Node=362623.4
       1    4970    5350
Encroach Node=361421.5
       1    4985    5285
Encroach Node=360650.7
       1    4700    5217
Encroach Node=359656.4
       1    4895    5260
Encroach Node=358871.8
       1    4915    5025
Encroach Node=358760
       1  4959.6  5049.5
Encroach Node=358711.9
       1  4959.6  5049.5
Encroach Node=358670
       1  4959.6  5049.5
Encroach Node=358431.6
       1    4955    5220
Encroach Node=357927.6
       1    4985    5280
Encroach Node=356334.4
       1    4530    5060
Encroach Node=355818.6
       1    4560    5015
Encroach Node=355803.6
       1    4560    5015
Encroach Node=355788.6
       1    4560    5015
Encroach Node=355220.5
       1    4850    5305
Encroach Node=354502.3
       1    4610    5020
Encroach Node=353146.4
       1    4380    5020
Encroach Node=352519.9
       1    4865    5485
Encroach Node=352448.5
       1    4895    5520
Encroach Node=352431.5
       1    4895    5520
Encroach Node=352414.5
       1    4895    5520
Encroach Node=352094.8
       1    4730    5480
Encroach Node=351184.1
       1    4700    5195
Encroach Node=349666.6
       1    4980    5715
Encroach Node=348410.9
       1    4525    5020
Encroach Node=347486.7
       1    4964    5614
Encroach Node=346570.3
       1    4650    5020
Encroach Node=344901.6
       1    4368    5073
Encroach Node=343432.7
       1    4520    5016
Encroach Node=342134.8
       1    4779    5340
Encroach Node=341654.0
       1    4875    5345
Encroach Node=340883.3
       1    4455    5045
Encroach Node=340800.4
       1    4455    5300
Encroach Node=340768.9
       1    4455    5300
Encroach Node=340737.4
       1    4455    5300
Encroach Node=340480.0
       1    4590    5365
Encroach Node=339806.4
       1    4510    5395
Encroach Node=338783.3
       1    4810    5490
Encroach Node=337922.3
       1    4067    5021
Encroach Node=337168.3
       1    3813    5058
Encroach Node=335710.7
       1    4000    5240
Encroach Node=333741.8
       1    4400    5020
Encroach Node=333114.7
       1    4255    5025
Encroach Node=332505.1
       1    3865    5015
Encroach Node=332186.3
       1    3945    5050
Encroach Node=331980.1
       1    3950    5050
Encroach Node=331810
       1    3920    5030
Encroach Node=331768
       1    3920    5030
Encroach Node=331726
       1    3920    5030
Encroach Node=331580.1
       1    3875    5040
Encroach Node=331161.5
       1    3850    5170
Encroach Node=329870.1
       1    4645    5700
Encroach Node=329103.9
       1    4622    5593
Encroach Node=327680.9
       1    3920    5075
Encroach Node=326067.5
       1    4980    5870
Encroach Node=324978.2
       1    4735    5510
Encroach Node=324699.3
       1    4640    5395
Encroach Node=324675.3
       1    4640    5395
Encroach Node=324651.3
       1    4640    5395
Encroach Node=324448.5
       1    4665    5430
Encroach Node=324126.4
       1    4710    5450
Encroach Node=322581.7
       1    4930    6005
Encroach Node=322049.6
       1    4980    5510
Encroach Node=320841.0
       1    4678    5163
Encroach Node=319539.7
       1    4980    5305
Encroach Node=318256.3
       1    4699    5249
Encroach Node=317377.2
       1    4980    5435
Encroach Node=316442.7
       1    4680    5790
Encroach Node=314695.6
       1    4555    5035
Encroach Node=314083.9
       1    4530    5075
Encroach Node=313747.7
       1    4630    5080
Encroach Node=313556.0
       1    4530    5060
Encroach Node=313528.0
       1    4530    5060
Encroach Node=313500.0
       1    4530    5060
Encroach Node=313379.2
       1    4485    5030
Encroach Node=312917.5
       1    4560    5040
Encroach Node=312109.2
       1    4450    5170
Encroach Node=310620.7
       1    4740    5080
Encroach Node=309811.2
       1    4628    5032
Encroach Node=308858.1
       1    4975    5335
Encroach Node=308143.7
       1    4159    5066
Encroach Node=307032.4
       1    4885    5430
Encroach Node=306637.5
       1    4935    5240
Encroach Node=305929.2
       1    4855    5240
Encroach Node=305093.2
       1    4925    5280
Encroach Node=304581.5
       1    4840    5200
Encroach Node=303924.9
       1    4843    5145
Encroach Node=303573.5
       1    4880    5200
Encroach Node=303021.8
       1    4674    5116
Encroach Node=301168.9
       1    4700    5110
Encroach Node=300789.3
       1    4650    5430
Encroach Node=300588.4
       1    4290    5080
Encroach Node=300563.4
       1    4290    5080
Encroach Node=300538.4
       1    4290    5080
Encroach Node=300417.1
       1    4600    5450
Encroach Node=300206.7
       1    4600    5450
Encroach Node=299727.1
       1    4495    5425
Encroach Node=298613.9
       1    4235    5020
Encroach Node=296972.1
       1    4930    5370
Encroach Node=295216.8
       1  3673.5    5095
Encroach Node=293785.3
       1    4265    5040
Encroach Node=292719.4
       1    4500    5240
Encroach Node=291773.9
       1    4800    5365
Encroach Node=290617.0
       1    4370    5010
Encroach Node=289038.3
       1    4977    5630
Encroach Node=288387.2
       1    4910    5535
Encroach Node=288254.7
       1    4880    5595
Encroach Node=288228.7
       1    4880    5595
Encroach Node=288202.7
       1    4880    5595
Encroach Node=288101.9
       1    4820    5500
Encroach Node=287629.8
       1    4808    5451
Encroach Node=286810.8
       1    4340    5025
Encroach Node=286019.2
       1    4780    5390
Encroach Node=285474.5
       1    4820    5505
Encroach Node=284884.7
       1    4840    5425
Encroach Node=284224.5
       1    4779    5414
Encroach Node=283056.7
       1    4560    5135
Encroach Node=281683.2
       1    4250    5150
Encroach Node=281325.9
       1    4000    5350
Encroach Node=281309.9
       1    4000    5350
Encroach Node=281293.9
       1    4000    5350
Encroach Node=281230.1
       1    4000    5400
Encroach Node=280415.4
       1    4300    5240
Encroach Node=279957.0
       1    4685    5420
Encroach Node=278974.0
       1    4205    5500
Encroach Node=276574.0
       1    4570    6110
Encroach Node=275250.8
       1    4410    5460
Encroach Node=274419.1
       1    4725    5555
Encroach Node=273050.2
       1    4619    5165
Encroach Node=271847.4
       1    4401    5024
Encroach Node=270264.8
       1    4550    5566
Encroach Node=268978.8
       1    4113    5057
Encroach Node=268443.6
       1    4259    5069
Encroach Node=267069.3
       1    4922    5663
Encroach Node=266006.8
       1    4578    5564
Encroach Node=265776.4
       1    4555    5485
Encroach Node=265745.1
       1    4555    5485
Encroach Node=265713.9
       1    4555    5485
Encroach Node=265483.0
       1    4301    5381
Encroach Node=265026.2
       1    4002    5048
Encroach Node=264692.5
       1    3930    5078
Encroach Node=263211.6
       1    4511    5441
Encroach Node=262727.2
       1    4703    5487
Encroach Node=261953.2
       1    4380    5158
Encroach Node=260953.0
       1    4885    5411
Encroach Node=260773.2
       1    4930    5439
Encroach Node=260537.4
       1    4935    5441
Encroach Node=260505.9
       1    4935    5441
Encroach Node=260474.4
       1    4935    5441
Encroach Node=260390.6
       1    4850    5392
Encroach Node=260014.0
       1    4683    5178
Encroach Node=259563.8
       1    4582    5040
Encroach Node=258009.9
       1    4403    5554
Encroach Node=257100.6
       1    4170    5163
Encroach Node=255371.0
       1    4707    5568
Encroach Node=254627.6
       1    4925    5615
Encroach Node=253915.9
       1    4400    5376
Encroach Node=253565.0
       1    4095    5200
Encroach Node=253257.0
       1    3850    5065
Encroach Node=253220.0
       1    3850    5065
Encroach Node=253183.0
       1    3850    5065
Encroach Node=253055.3
       1    3593    5065
Encroach Node=252295.8
       1    3640    5175
Encroach Node=250563.3
       1    3945    5450
Encroach Node=249516.8
       1    4125    5565
Encroach Node=247895.6
       1    4704    6150
Encroach Node=246746.6
       1    4580    5835
Encroach Node=244790.2
       1    4350    5600
Encroach Node=243422.6
       1    3846    5136
Encroach Node=242215.8
       1    4830    6150
Encroach Node=241149.2
       1    4870    6150
Encroach Node=239561.0
       1  4272.2    5290
Encroach Node=239260.1
       1    4080    5160
Encroach Node=239229.6
       1    4080    5160
Encroach Node=239199.1
       1    4080    5160
Encroach Node=238748.0
       1    3918    5069
Encroach Node=237861.9
       1    4000    5200
Encroach Node=236547.8
       1    4056    5305
Encroach Node=235332.5
       1    3390    5080
Encroach Node=234734.7
       1    3370  5041.8
Encroach Node=233292.2
       1    3270    5680
Encroach Node=230694.7
       1    3803    6925
Encroach Node=229710.8
       1    4065    6745
Encroach Node=228588.3
       1    3640    6025
Encroach Node=227253.1
       1    2250    5297
Encroach Node=225153.4
       1    1305    5040
Encroach Node=223808.7
       1    1390    5155
Encroach Node=221840.8
       1    2832    6385
Encroach Node=221103.6
       1    3400    6230
Encroach Node=219902.0
       1    3450    5515
Encroach Node=217354.5
       1  4309.8  6359.3
Encroach Node=213918.9
       1    2740    5200
Encroach Node=211631.6
       1    3300    5250
Encroach Node=210431.1
       1    3850    5600
Encroach Node=209190.3
       1    4260    5905
Encroach Node=208249.9
       1    4510    6005
Encroach Node=207799.6
       1  4212.5    6065
Encroach Node=207518.1
       1    3650    5900
Encroach Node=207453.1
       1    3650    5900
Encroach Node=207388.1
       1    3650    5900
Encroach Node=207139.4
       1    3621    5800
Encroach Node=206325.6
       1    2745    5415
Encroach Node=205172.3
       1    2980    5140
Encroach Node=203889.5
       1    3515    5380
Encroach Node=202317.6
       1    3770    6170
Encroach Node=201301.7
       1    2835    5625
Encroach Node=199974.4
       1    2795    5040
Encroach Node=198833.4
       1    3575    5320
Encroach Node=198488.0
       1    3850    5300
Encroach Node=198318.6
       1    3850  5165.9
Encroach Node=198300.6
       1    3850  5165.9
Encroach Node=198282.6
       1    3850  5165.9
Encroach Node=198097.0
       1    3860    5450
Encroach Node=196302.3
       1    2625    5060
Encroach Node=193888.1
       1    3770    5550
Encroach Node=192987.0
       1    4300    6125
Encroach Node=192144.6
       1    4515    6480
Encroach Node=191675.8
       1    4664    6373
Encroach Node=190756.0
       1    4150  5325.7
Encroach Node=190739.5
       1    4150  5325.7
Encroach Node=190723.0
       1    4150  5325.7
Encroach Node=189712.6
       1    3950    5035
Encroach Node=188775.6
       1    3650    5090
Encroach Node=187576.7
       1    3250    5255
Encroach Node=186599.3
       1    4065    5600
Encroach Node=184626.4
       1    3085    5600
Encroach Node=182543.1
       1    3062    5030
Encroach Node=181868.6
       1    3700    5300
Encroach Node=181706.6
       1    3733    5385
Encroach Node=181671.6
       1    3733    5385
Encroach Node=181636.6
       1    3733    5385
Encroach Node=181281.7
       1    3500    5100
Encroach Node=180714.4
       1    3565    5280
Encroach Node=179254.7
       1    3330    5225
Encroach Node=177593.4
       1    3135    5085
Encroach Node=176206.0
       1    3257    5035
Encroach Node=174131.0
       1    3400    5495
Encroach Node=172966.9
       1    4280    6525
Encroach Node=171768.5
       1    4390    6731
Encroach Node=170367.7
       1    4460    7238
Encroach Node=168865.4
       1    4785    7475
Encroach Node=165536.3
       1    4743    7645
Encroach Node=163482.3
       1    4750    8040
Encroach Node=162164.1
       1    3850    7390
Encroach Node=159174.0
       1    2000    5617
Encroach Node=157651.2
       1    1975    5105
Encroach Node=156001.8
       1    3303    5340
Encroach Node=155042.3
       1    3070    5710
Encroach Node=153682.2
       1    4285    6670
Encroach Node=153142.6
       1    4175    6765
Encroach Node=151553.1
       1    3660    6400
Encroach Node=150642.0
       1    3335    5690
Encroach Node=149311.7
       1    4450    6195
Encroach Node=148935.1
       1    4629    6215
Encroach Node=148908.1
       1    4629    6105
Encroach Node=148881.1
       1    4629    5975
Encroach Node=148606.0
       1    4450    5960
Encroach Node=147849.6
       1    3700    5640
Encroach Node=146208.1
       1    3766    5560
Encroach Node=144510.7
       1    3335    5435
Encroach Node=141923.5
       1    4030    6036
Encroach Node=140963.4
       1    4080    6050
Encroach Node=139160.1
       1    3190    5320
Encroach Node=137656.0
       1    2675    5670
Encroach Node=136198.2
       1    3985    6045
Encroach Node=135401.0
       1    3850    5504
Encroach Node=134528.2
       1    4470    6125
Encroach Node=133785.6
       1    4215    5905
Encroach Node=131665.9
       1    4800    6125
Encroach Node=130131.1
       1    4315    6270
Encroach Node=129178.8
       1    4175    5765
Encroach Node=128719.4
       1 3983.69    5775
Encroach Node=128687.4
       1 3983.69    5775
Encroach Node=128636.7
       1 3983.69    5775
Encroach Node=128210.0
       1    4105    5675
Encroach Node=127566.0
       1    4190    6710
Encroach Node=126725.2
       1    3725    6475
Encroach Node=125593.6
       1    3675    6135
Encroach Node=124486.4
       1    3500  6432.1
Encroach Node=122390.6
       1    4160    6960
Encroach Node=121286.5
       1    4834    6950
Encroach Node=120290.5
       1    4345    6440
Encroach Node=117085.2
       1 3361.83 5283.16
Encroach Node=115715.2
       1  3635.6  5211.5
Encroach Node=114331.8
       1  3793.6 5384.76
Encroach Node=112909.9
       1 4506.63 5627.23
Encroach Node=110554.7
       1    3790    5850
Encroach Node=109165.1
       1    3530    5590
Encroach Node=107034.5
       1    3900    5875
Encroach Node=106148.0
       1    4300    6250
Encroach Node=104333.5
       1    3580    5880
Encroach Node=102794.9
       1    3770    5565
Encroach Node=100852.5
       1    3230    5120
Encroach Node=100361.0
       1    3092    5070
Encroach Node=99039.0
       1    3695    5649
Encroach Node=97170.6
       1    3720    6490
Encroach Node=95303.6
       1    3270    5940
Encroach Node=94465.9
       1  2717.4    5175
Encroach Node=93038.3
       1    3620    5310
Encroach Node=91780.8
       1    4275    5996
Encroach Node=90249.3
       1    4030    5750
Encroach Node=88797.0
       1    3575    5805
Encroach Node=88153.2
       1    3855    5790
Encroach Node=87559.3
       1    4055    5870
Encroach Node=87195.6
       1    3290    4835
Encroach Node=86927.5
       1    3290    4835
Encroach Node=86681.8
       1    3290    4835
Encroach Node=85856.6
       1    3745    5660
Encroach Node=84744.7
       1    3420    5890
Encroach Node=83099.6
       1    4160    6775
Encroach Node=82761.5
       1    4470    6975
Encroach Node=82743.3
       1    4470    6975
Encroach Node=82725.2
       1    4470    6975
Encroach Node=82073.8
       1    4765    7076
Encroach Node=80878.1
       1    4635    6495
Encroach Node=79447.2
       1    4225    6280
Encroach Node=78116.0
       1    3600    6705
Encroach Node=76553.3
       1    3170    5070
Encroach Node=76082.3
       1    3327    5070
Encroach Node=75018.5
       1    3780    5650
Encroach Node=73296.0
       1    4132    7019
Encroach Node=72547.7
       1    4786    6625
Encroach Node=71829.0
       1    4207    5813
Encroach Node=71348.7
       1    4150    5575
Encroach Node=70767.1
       1    4490    6035
Encroach Node=69737.8
       1    3580    5510
Encroach Node=69232.2
       1    3960    5760
Encroach Node=68984.0
       1    4110    5259
Encroach Node=68728.6
       1    3574    5362
Encroach Node=68706.1
       1    3574    5362
Encroach Node=68683.6
       1    3574    5362
Encroach Node=68507.9
       1    3640    5385
Encroach Node=68065.2
       1    3630    5750
Encroach Node=67818.7
       1    3660    5940
Encroach Node=67196.3
       1    3350    6200
Encroach Node=65844.4
       1    3110    6080
Encroach Node=64135.5
       1    2850    5505
Encroach Node=62959.6
       1    2618    5766
Encroach Node=61564.3
       1    2788    5810
Encroach Node=60210.3
       1    3540    5455
Encroach Node=58691.8
       1    4770    6500
Encroach Node=57733.4
       1    4625    6320
Encroach Node=56314.1
       1    4350    6545
Encroach Node=53962.3
       1    4680    6345
Encroach Node=52217.8
       1    4025    6625
Encroach Node=49773.6
       1    4153    5867
Encroach Node=48076.0
       1    4654    7162
Encroach Node=46243.5
       1    4430    6680
Encroach Node=45403.9
       1    4229    6445
Encroach Node=43924.4
       1    4625    6393
Encroach Node=42546.8
       1    3570    6190
Encroach Node=41576.1
       1    4300    6755
Encroach Node=40938.2
       1    4410    6900
Encroach Node=39313.9
       1    3340    6125
Encroach Node=36356.7
       1    2271    5100
Encroach Node=35047.8
       1    3450    5731
Encroach Node=34111.6
       1    3490    6110
Encroach Node=32535.7
       1    3000    5741
Encroach Node=31192.2
       1    2730    5440
Encroach Node=29692.8
       1    2500    5260
Encroach Node=29028.0
       1    2785    5070
Encroach Node=27592.1
       1    4500    5702
Encroach Node=26862.3
       1    4100    5585
Encroach Node=25883.5
       1    3100    5400
Encroach Node=24783.7
       1    2550    5315
Encroach Node=23405.3
       1    3045    5720
Encroach Node=22403.9
       1    4100    6030
Encroach Node=21505.6
       1    3750    5810
Encroach Node=20617.2
       1    3520    5865
Encroach Node=19133.4
       1    2917    6412
Encroach Node=17516.9
       1    3000    5520
Encroach Node=16413.7
       1    2390    5700
Encroach Node=15655.4
       1    2030    5254
Encroach Node=14080.8
       1    3320    6235
Encroach Node=13076.9
       1    3595    6120
Encroach Node=12248.6
       1    3635    6250
Encroach Node=10706.6
       1    4860    6550
Encroach Node=9272.5
       1  4365.5  5920.5
Encroach Node=8103.2
       1    4824    5692
Encroach Node=6876.4
       1    4684    5549
Encroach Node=5239.9
       1    3693    5372
Encroach Node=3019.7
       1    3557    6085
BEGIN DESCRIPTION:
FEMA Effective June 2007 +...+ LOMR 14-06-1656P
END DESCRIPTION:
Computation Interval=1HOUR
Output Interval=1HOUR
Run HTab= 0
Run UNet= 0
Run PostProcess= 0
UNET Theta= 1
UNET ZTol= 0.02
UNET ZSATol= 0.1
UNET MxIter= 20
UNET MaxInSteps= 20
UNET DtIC= 0
UNET DtMin= 0
UNET MaxCRTS= 20
UNET WFStab= 2
UNET SFStab= 1
UNET WFX= 1
UNET SFX= 1
UNET Convert EG Bridges=-1
UNET Use Existing IB Tables=-1
Instantaneous Interval=1HOUR
Write IC File= 0
Write Velocity= 0
Write Detailed= 0

--- J100-00-00.f01 (steady flow) ---

Flow Title=FEMA Effective June 2007
Version=Version 3.0.1  Mar 2001
Number of Profiles= 4
Profile Names=10PCT_10yr, 2PCT_50yr, 1PCT_100yr, 0.2PCT_500yr
River Rch & RM=J100-00-00,J100-00-00_0030,367736.2
     510     890    1100    1700
River Rch & RM=J100-00-00,J100-00-00_0030,366583.5
     550     950    1200    1800
River Rch & RM=J100-00-00,J100-00-00_0030,365737.8
     600    1000    1300    2000
River Rch & RM=J100-00-00,J100-00-00_0030,364609.2
     700    1200    1600    2400
River Rch & RM=J100-00-00,J100-00-00_0030,362623.4
     800    1400    1900    2900
River Rch & RM=J100-00-00,J100-00-00_0030,360650.7
    1000    1700    2200    3500
River Rch & RM=J100-00-00,J100-00-00_0030,358760
    1200    2000    2500    4000
River Rch & RM=J100-00-00,J100-00-00_0030,356334.4
    1400    2300    2800    4500
River Rch & RM=J100-00-00,J100-00-00_0030,354502.3
    1500    2500    3100    4900
River Rch & RM=J100-00-00,J100-00-00_0030,353146.4
    1600    2600    3200    5100
River Rch & RM=J100-00-00,J100-00-00_0030,352519.9
    1700    2700    3300    5300
River Rch & RM=J100-00-00,J100-00-00_0030,351184.1
    1900    3000    3800    6000
River Rch & RM=J100-00-00,J100-00-00_0030,347486.7
    2000    3300    4100    6600
River Rch & RM=J100-00-00,J100-00-00_0030,344901.6
    2000    3400    4200    6700
River Rch & RM=J100-00-00,J100-00-00_0030,343432.7
    2136    3698    4542    7041
River Rch & RM=J100-00-00,J100-00-00_0030,340480
    2200    3800    4700    7300
River Rch & RM=J100-00-00,J100-00-00_0030,337168.3
    2300    4000    4900    7800
River Rch & RM=J100-00-00,J100-00-00_0030,332505.1
    2400    4200    5200    8200
River Rch & RM=J100-00-00,J100-00-00_0030,327680.9
    2400    4300    5300    8500
River Rch & RM=J100-00-00,J100-00-00_0030,324978.2
    2500    4400    5500    8900
River Rch & RM=J100-00-00,J100-00-00_0030,320841
    2500    4600    5700    9300
River Rch & RM=J100-00-00,J100-00-00_0030,317377.2
    2600    4700    5900    9600
River Rch & RM=J100-00-00,J100-00-00_0030,314695.6
    2700    4800    6100    9900
River Rch & RM=J100-00-00,J100-00-00_0030,312109.2
    2700    4900    6200   10200
River Rch & RM=J100-00-00,J100-00-00_0030,309811.2
    2700    5000    6300   10400
River Rch & RM=J100-00-00,J100-00-00_0030,308143.7
    2800    5200    6500   10900
River Rch & RM=J100-00-00,J100-00-00_0030,304581.5
    2892    5353    6804   11414
River Rch & RM=J100-00-00,J100-00-00_0030,300588.4
    3800    7000    9000   15500
River Rch & RM=J100-00-00,J100-00-00_0030,296972.1
    3900    7300    9400   16100
River Rch & RM=J100-00-00,J100-00-00_0030,290617
    4100    7600    9800   16700
River Rch & RM=J100-00-00,J100-00-00_0030,284224.5
    4300    7800   10000   17200
River Rch & RM=J100-00-00,J100-00-00_0030,279957
    4500    8300   10600   18100
River Rch & RM=J100-00-00,J100-00-00_0030,271847.4
    4700    8700   11100   18800
River Rch & RM=J100-00-00,J100-00-00_0030,265026.2
    4900    8900   11300   19200
River Rch & RM=J100-00-00,J100-00-00_0030,261953.2
    4949    9030   11503   19487
River Rch & RM=J100-00-00,J100-00-00_0030,258009.9
   11510   20900   26167   43073
River Rch & RM=J100-00-00,J100-00-00_0030,229710.8
   16919   34150   44311   74666
River Rch & RM=J100-00-00,J100-00-00_0030,188775.6
   23039   43568   54003   87322
River Rch & RM=J100-00-00,J100-00-00_0030,155042.3
   22888   43509   54138   87983
River Rch & RM=J100-00-00,J100-00-00_0030,133785.6
   22460   42884   49790   67233
River Rch & RM=J100-00-00,J100-00-00_0030,110554.7
   24485   46922   54599   78875
River Rch & RM=J100-00-00,J100-00-00_0030,93038.3
   23336   45957   57889  102286
River Rch & RM=J100-00-00,J100-00-00_0030,68728.6
   22890   45287   57345  101084
River Rch & RM=J100-00-00,J100-00-00_0030,36356.7
   22579   44774   56871  100372
River Rch & RM=J100-00-00,J100-00-00_0030,19133.4
   30772   60592   76749  132093
Boundary for River Rch & Prof#=J100-00-00,J100-00-00_0030, 1
Up Type= 0
Dn Type= 1
Dn Known WS=58.1
Boundary for River Rch & Prof#=J100-00-00,J100-00-00_0030, 2
Up Type= 0
Dn Type= 1
Dn Known WS=64.8
Boundary for River Rch & Prof#=J100-00-00,J100-00-00_0030, 3
Up Type= 0
Dn Type= 1
Dn Known WS=67.1
Boundary for River Rch & Prof#=J100-00-00,J100-00-00_0030, 4
Up Type= 0
Dn Type= 1
Dn Known WS=73.8
DSS Import GetInterval= 0
DSS Import GetPeak= 0
DSS Import FillOption= 0

--- J100-00-00.f02 (steady flow) ---

Flow Title=Floodway
Version=Version 3.0.1  Mar 2001
Number of Profiles= 2
Profile Names=11PCT_100yr, 1PCTFloodway_100yrFW
River Rch & RM=J100-00-00,J100-00-00_0030,367736.2
    1100    1100
River Rch & RM=J100-00-00,J100-00-00_0030,366583.5
    1200    1200
River Rch & RM=J100-00-00,J100-00-00_0030,365737.8
    1300    1300
River Rch & RM=J100-00-00,J100-00-00_0030,364609.2
    1600    1600
River Rch & RM=J100-00-00,J100-00-00_0030,362623.4
    1900    1900
River Rch & RM=J100-00-00,J100-00-00_0030,360650.7
    2200    2200
River Rch & RM=J100-00-00,J100-00-00_0030,358760
    2500    2500
River Rch & RM=J100-00-00,J100-00-00_0030,356334.4
    2800    2800
River Rch & RM=J100-00-00,J100-00-00_0030,354502.3
    3100    3100
River Rch & RM=J100-00-00,J100-00-00_0030,353146.4
    3200    3200
River Rch & RM=J100-00-00,J100-00-00_0030,352519.9
    3300    3300
River Rch & RM=J100-00-00,J100-00-00_0030,351184.1
    3800    3800
River Rch & RM=J100-00-00,J100-00-00_0030,347486.7
    4100    4100
River Rch & RM=J100-00-00,J100-00-00_0030,344901.6
    4200    4200
River Rch & RM=J100-00-00,J100-00-00_0030,343432.7
    4542    4542
River Rch & RM=J100-00-00,J100-00-00_0030,340480
    4700    4700
River Rch & RM=J100-00-00,J100-00-00_0030,337168.3
    4900    4900
River Rch & RM=J100-00-00,J100-00-00_0030,332505.1
    5200    5200
River Rch & RM=J100-00-00,J100-00-00_0030,327680.9
    5300    5300
River Rch & RM=J100-00-00,J100-00-00_0030,324978.2
    5500    5500
River Rch & RM=J100-00-00,J100-00-00_0030,320841
    5700    5700
River Rch & RM=J100-00-00,J100-00-00_0030,317377.2
    5900    5900
River Rch & RM=J100-00-00,J100-00-00_0030,314695.6
    6100    6100
River Rch & RM=J100-00-00,J100-00-00_0030,312109.2
    6200    6200
River Rch & RM=J100-00-00,J100-00-00_0030,309811.2
    6300    6300
River Rch & RM=J100-00-00,J100-00-00_0030,308143.7
    6500    6500
River Rch & RM=J100-00-00,J100-00-00_0030,304581.5
    6804    6804
River Rch & RM=J100-00-00,J100-00-00_0030,300588.4
    9000    9000
River Rch & RM=J100-00-00,J100-00-00_0030,296972.1
    9400    9400
River Rch & RM=J100-00-00,J100-00-00_0030,290617
    9800    9800
River Rch & RM=J100-00-00,J100-00-00_0030,284224.5
   10000   10000
River Rch & RM=J100-00-00,J100-00-00_0030,279957
   10600   10600
River Rch & RM=J100-00-00,J100-00-00_0030,271847.4
   11100   11100
River Rch & RM=J100-00-00,J100-00-00_0030,265026.2
   11300   11300
River Rch & RM=J100-00-00,J100-00-00_0030,261953.2
   11503   11503
River Rch & RM=J100-00-00,J100-00-00_0030,258009.9
   26167   26167
River Rch & RM=J100-00-00,J100-00-00_0030,229710.8
   44311   44311
River Rch & RM=J100-00-00,J100-00-00_0030,188775.6
   54003   54003
River Rch & RM=J100-00-00,J100-00-00_0030,155042.3
   54138   54138
River Rch & RM=J100-00-00,J100-00-00_0030,133785.6
   49790   49790
River Rch & RM=J100-00-00,J100-00-00_0030,110554.7
   54599   54599
River Rch & RM=J100-00-00,J100-00-00_0030,93038.3
   57889   57889
River Rch & RM=J100-00-00,J100-00-00_0030,68728.6
   57345   57345
River Rch & RM=J100-00-00,J100-00-00_0030,36356.7
   56871   56871
River Rch & RM=J100-00-00,J100-00-00_0030,19133.4
   76749   76749
Boundary for River Rch & Prof#=J100-00-00,J100-00-00_0030, 1
Up Type= 0
Dn Type= 1
Dn Known WS=67.1
Boundary for River Rch & Prof#=J100-00-00,J100-00-00_0030, 2
Up Type= 0
Dn Type= 1
Dn Known WS=68.1
DSS Import GetInterval= 0
DSS Import GetPeak= 0
DSS Import FillOption= 0

--- J100-00-00.g01 (geometry) ---

Geom Title=J100-00-00
Version=Version 3.0.1  May 2012

River Reach=J100-00-00      ,J100-00-00_0030
Reach XY= 30
    2928911.1445   13983101.5741    2948756.0895   13968139.5814
    2956853.7586   13968718.3303    2960660.0905   13962839.9861
    2965605.4417   13961113.3951    2968130.0087    13954948.996
    2975072.5086   13954584.4612    2983812.6896   13959534.6242
    2992578.3794    13956571.885    3007223.5844   13963009.2272
    3014917.0096   13961910.6339    3016854.9685   13965049.5103
    3021794.2514    13963075.524    3031602.1485   13972511.5714
    3035811.6595   13972796.9392    3035830.8784   13975975.6062
    3046279.4807   13976282.2865       3057783.5       13989174.
     3061074.956   13989320.1394    3074610.0783    13979625.644
    3078777.1414    13967037.651    3089340.4902   13966093.5679
    3098874.6547   13970437.9342    3107533.6494   13959698.7899
    3115019.5416   13960294.0141    3115879.7847   13957553.5627
    3122731.3472   13956968.4932    3133790.1391    13949187.518
    3137347.2326   13940444.1877        3150683.       13941807.
